HEC-RAS study LtlGraveCk.prj: LtlGraveCk

--- LtlGraveCk.g01 (geometry) --- (continued)

Type RM Length L Ch R = 1 ,19187   ,295.4,299.8,295.7
XS GIS Cut Line= 6
1632147.47080925534244.9905345891632111.37737751 534324.65212068
1632080.43911918534392.9370890861632038.81584284534483.915581673
1632002.27457733534550.048651502  1631957.867842 534627.93891567
#Sta/Elev= 30
       0  882.92     4.5  881.67    11.2  878.34    43.6  851.36    46.6  849.23
      58  842.75    61.6  841.51    78.9  838.65   101.2  836.19   108.6  835.75
   150.7  834.43   196.2  834.45   198.5  834.14   200.3  833.29  205.32829.7732
   209.3  828.09   212.6  827.93   217.6   828.3  227.41829.7715   237.4  831.32
     267  833.12   297.2  833.55   304.7  834.23   323.5  833.88   342.2  834.12
   368.7  836.32   372.5   836.8   380.3  838.74   417.8  850.03   427.7  851.66
#Mann= 5, -1 ,  0
       0     0.1       0  205.32   0.045       0  227.41     0.1       0
  232.42    0.06       0  408.03    0.05       0
Bank Sta=205.32,227.41
XS Rating Curve= 0 ,0
Exp/Cntr(USF)=0,0
Exp/Cntr=0.3,0.1

Type RM Length L Ch R = 1 ,18887   ,322.7,324,324.6
XS GIS Cut Line= 6
1631883.77743901534171.7072165911631850.44056343534254.699504673
1631813.11091368534319.7571173461631762.17597617534405.813375667
  1631723.974609534470.3552413431631679.33821534534545.604762763
#Sta/Elev= 30
       0  865.28    15.7  853.33    24.7  842.44    29.8  837.46    33.4  835.42
    36.9  834.59      65  832.07   112.7  830.58   135.9  830.85   162.3  832.49
   184.7  830.13   196.1  829.79   199.9   828.8  204.22825.9921   207.6  824.53
   214.7  824.21     219  824.29  223.86825.9889   230.4  829.36   234.3  829.97
   241.9  829.68   253.3   830.5     280  829.78   314.3  831.36   337.2  837.25
   363.9  846.68     395  850.55   401.8  852.41   413.8  857.21   426.9  860.85
#Mann= 5, -1 ,  0
       0     0.1       0  119.44    0.06       0  204.22   0.045       0
  223.86    0.06       0  324.44    0.05       0
Bank Sta=204.22,223.86
XS Rating Curve= 0 ,0
Exp/Cntr(USF)=0,0
Exp/Cntr=0.3,0.1

Type RM Length L Ch R = 1 ,18563   ,276.5,276,274.5
XS GIS Cut Line= 2
1631652.00645884534005.0073002091631400.96016318534342.749197334
#Sta/Elev= 30
       0  889.33     9.2  885.29      21  882.24    31.3  877.97    47.8  875.09
    58.8  871.33    64.3  868.82    70.5  865.29    74.6  862.35    86.3  851.19
    99.1  840.75   105.4  836.33   111.4  833.48   156.4  828.16     185  826.88
   189.1  825.72  193.67823.0432   197.2  821.62   205.4  821.18   210.9  821.59
  215.89823.0409   222.6  824.81   240.3   826.9   255.5  826.71   262.6   827.6
     279  827.75   295.3  828.91   323.5  831.47     373   837.2   420.8  841.03
#Mann= 5, -1 ,  0
       0     0.1       0     150    0.06       0  193.67   0.045       0
  215.89    0.06       0     420    0.05       0
Bank Sta=193.67,215.89
XS Rating Curve= 0 ,0
Exp/Cntr(USF)=0,0
Exp/Cntr=0.3,0.1

Type RM Length L Ch R = 1 ,18287   ,378.9,378.3,377.4
XS GIS Cut Line= 6
1631405.27216242533844.8459936681631360.75519109533920.180816755
1631322.59581859533984.7587715831631271.61494942534070.787470922
1631231.73510793534134.3263858411631183.17155676534207.258982763
#Sta/Elev= 30
       0  910.85     7.9  909.84    19.3  906.45    38.4  897.99      46   895.2
    53.6  892.78    72.7  888.16    76.5  885.99    91.7  871.54   116.3  852.39
     126     844   129.8  841.51   154.6  828.03   160.3  826.18   167.9  825.11
     187  824.09   194.6  823.18  202.07820.9758   207.3  819.37   213.7  819.04
   221.3  819.66  224.49820.9767   228.9  823.43   233.7   824.5   264.8  824.96
   325.3  827.64   341.1  829.34   376.3  834.12   404.8  836.54   425.2  837.56
#Mann= 6, -1 ,  0
       0     0.1       0   157.5    0.06       0  202.07   0.045       0
  224.49    0.06       0  397.53    0.05       0  417.53    0.06       0
Bank Sta=202.07,224.49
XS Rating Curve= 0 ,0
Exp/Cntr(USF)=0,0
Exp/Cntr=0.3,0.1

Type RM Length L Ch R = 1 ,17909   ,205.3,207.3,208.5
XS GIS Cut Line= 2
1631058.92073424533664.7644100221630864.92517941 534044.90326474
#Sta/Elev= 30
       0  890.37    19.2  883.91      33  880.83    47.7  875.73    69.8  871.37
    77.2  869.36    84.6   866.4    92.4  861.74    95.6  860.78     103  860.16
   111.9  856.64   121.6  853.85   139.8  846.26   154.5  841.39   172.9  833.47
   180.2   829.3   187.1  824.34  194.54817.8328   198.7  816.38   202.4   816.2
   213.5  816.58  217.73817.8353   224.1  819.98   228.2   820.4   305.5  821.54
   320.3  822.46   341.1  827.62   357.1  834.18   368.2  837.77   426.8  845.46
#Mann= 4, -1 ,  0
       0     0.1       0     110    0.06       0  194.54   0.045       0
  217.73    0.06       0
Bank Sta=194.54,217.73
XS Rating Curve= 0 ,0
Exp/Cntr(USF)=0,0
Exp/Cntr=0.3,0.1

Type RM Length L Ch R = 1 ,17702   ,314.5,322.5,333.1
XS GIS Cut Line= 2
1630926.23223104533559.1646664921630653.49315417533927.954423249
#Sta/Elev= 30
       0   868.7    19.2  857.52    48.4   847.2    57.8  841.58    62.4  839.55
    74.4  836.48    98.5  828.66   118.9  824.82   130.5  820.58   139.3  819.56
   167.9  818.88   224.3  819.42   228.9  818.48  234.68815.3728   239.9  813.93
   245.4  813.66   250.9  814.09  254.86815.3745   261.7  818.82   265.8  819.28
     327  819.99   361.3  822.23   367.4  823.07   384.1     827   396.4  828.86
   408.6     836   420.9  842.51   428.4  847.33   437.8  854.37   458.7  871.53
#Mann= 5, -1 ,  0
       0     0.1       0     210    0.06       0  234.68   0.045       0
  254.86    0.06       0     410     0.1       0
Bank Sta=234.68,254.86
XS Rating Curve= 0 ,0
Exp/Cntr(USF)=0,0
Exp/Cntr=0.3,0.1

Type RM Length L Ch R = 1 ,17379   ,58.8,58.8,57.5
XS GIS Cut Line= 4
1630897.95232532533502.1954665621630720.09794206533505.977861341
1630464.87894219533542.5916988691630375.67481217533636.944506586
#Sta/Elev= 30
       0  855.67    15.9  841.91    22.5  837.38    38.9  824.32    48.8  818.61
    55.3  816.52    65.2  816.03    81.6  817.09   120.1  816.45   230.1  817.68
   289.4  816.34   319.9  817.98   322.6  817.85   325.9  816.56  331.17812.8641
   339.1  810.94   352.4  811.55  356.65812.8666   365.6  819.95     369  820.65
   441.1  823.32   450.1  824.57   459.2  828.92   477.2  841.14   499.8  849.63
   513.4  855.74   522.4  857.74   535.9  863.28   544.9  865.85   565.6  869.38
#Mann= 5, -1 ,  0
       0     0.1       0     160    0.07       0  247.89    0.06       0
  331.17   0.045       0  356.65    0.06       0
Bank Sta=331.17,356.65
XS Rating Curve= 0 ,0
Exp/Cntr(USF)=0,0
Exp/Cntr=0.3,0.1

Type RM Length L Ch R = 1 ,17320   ,511.4,532,509.1
XS GIS Cut Line= 4
1630906.51483866533437.5524083791630648.58389423533452.354513411
1630443.32091417533493.3762350411630345.13776098533522.599380757
#Sta/Elev= 30
       0  864.66     8.1  856.78    14.7  851.36    24.5   840.9    27.8  838.58
    34.4  834.62    50.8  826.01    70.5  818.25    77.1  816.42   103.4  815.32
   159.3  815.43     179  815.89   192.1  815.19   211.9  814.99   241.1  813.41
   294.7  813.61   344.8  815.83   351.5  815.46   354.9  814.55  360.12812.4028
   364.9  811.21   371.6  810.82   381.6  811.09  386.09812.4048   388.2  813.58
     395   818.8   399.3  820.65   404.9  821.62   530.3  826.61   570.1   828.9
#Mann= 4, -1 ,  0
       0     0.1       0      80    0.06       0  360.12   0.045       0
  386.09    0.06       0
Bank Sta=360.12,386.09
XS Rating Curve= 0 ,0
Exp/Cntr(USF)=0,0
Exp/Cntr=0.3,0.1

Type RM Length L Ch R = 1 ,16788   ,365.1,366.5,344.2
XS GIS Cut Line= 3
1631000.42126609533167.594395429  1630913.413238533176.859140679
1630348.34207431533241.836132369
#Sta/Elev= 30
       0  934.66     6.9  926.81    16.8  919.36    40.5  909.54    53.1  906.49
    66.3  901.77    69.6  899.87    76.2  893.48    79.5  891.43    92.7  885.61
   119.1  864.45   145.5  837.86   165.3  821.15   178.5  815.95   195.1   812.4
  203.44807.0978   208.3  805.67   224.8  805.95  230.57807.0963   244.6  811.18
   290.8  812.85   343.7  811.52   432.8  812.06   475.8  812.58   545.1  815.42
   558.3  817.96   578.1  818.01   594.7  822.06   624.3  832.37   656.3  833.73
#Mann= 4, -1 ,  0
       0     0.1       0  203.44   0.045       0  230.57     0.1       0
   327.5    0.06       0
Bank Sta=203.44,230.57
XS Rating Curve= 0 ,0
Exp/Cntr(USF)=0,0
Exp/Cntr=0.3,0.1

Type RM Length L Ch R = 1 ,16422   ,227.7,233.7,237.2
XS GIS Cut Line= 3
1630724.36977254532777.993080806 1630520.8268763532999.134784968
1630338.97359445533146.156415457
#Sta/Elev= 30
       0  903.05     9.4  898.76      26   893.6    38.5  887.33    56.2  880.02
    65.5  875.22    72.4  869.88    94.7     846   101.5  840.29   137.4  818.05
   149.9  811.32   165.3  806.26  177.05803.4311   181.6  802.45   188.5  802.23
   207.1  802.42  213.82803.4307   222.6  806.16   225.7  806.53     242   806.6
   281.4  808.24   297.7  808.31   351.3  810.68   421.3  812.43   439.4   814.1
   460.5  814.47   494.2  817.81   498.5  818.76   518.9   825.8   534.4  829.48
#Mann= 5, -1 ,  0
       0     0.1       0  177.05   0.045       0  213.82    0.06       0
     240    0.07       0  370.56    0.06       0
Bank Sta=177.05,213.82
XS Rating Curve= 0 ,0
Exp/Cntr(USF)=0,0
Exp/Cntr=0.3,0.1

Type RM Length L Ch R = 1 ,16188   ,354.5,357.7,359.7
XS GIS Cut Line= 6
1630609.80984259532666.8463811731630537.54456717532717.265899763
 1630470.5853835532751.2084171771630380.55866067532794.850390255
1630314.77926467532832.894933596  1630239.528759532880.737685665
#Sta/Elev= 30
       0  879.25    12.2  874.04    20.1  869.56    26.3  864.05    48.1  840.85
    82.8  814.22    92.4  808.43    99.2  806.72   117.6  805.04   150.7  804.12
   183.6   804.1   187.8  803.42   194.5  801.16  203.05800.9296   212.8  799.45
   226.4  799.81  229.84800.9301   234.6  802.83   249.1  805.16   275.2  805.19
   286.6   806.6   297.9  809.78   316.9  809.86   339.6  818.83   360.7  821.01
   374.6  825.09   394.1  829.19   409.6  835.43   421.3  841.76   428.4  844.18
#Mann= 4, -1 ,  0
       0     0.1       0  203.05   0.045       0  229.84     0.1       0
  233.19    0.06       0
Bank Sta=203.05,229.84
XS Rating Curve= 0 ,0
Exp/Cntr(USF)=0,0
Exp/Cntr=0.3,0.1

Type RM Length L Ch R = 1 ,15831   ,278.5,280.4,281
XS GIS Cut Line= 6
1630485.57968596532411.0940607731630401.99848829532437.323667103
1630329.44581188532456.3269099391630232.70880063 532481.66380153
 1630160.1564523532500.6677005241630075.51193655532522.837931776
#Sta/Elev= 30
       0  870.23     5.9  867.36    29.4  852.44    41.8  849.39    55.6  841.84
    92.4   827.5   106.9  817.92   117.1  812.65   130.6  803.78   140.8   799.4
   146.1  798.88     173  800.27   198.5  800.23   218.8  798.51   232.4  800.59
  247.31796.8793   252.7  795.64   269.6  795.56  275.81796.8788   282.9  801.32
   286.6  802.15   310.4  803.53   330.7  815.32   336.9  817.91   344.3  819.69
   357.9  820.16   366.1  821.69   381.6     827   395.2   834.4   425.1  842.63
#Mann= 5, -1 ,  0
       0     0.1       0   232.6    0.06       0  247.31   0.045       0
  275.81    0.06       0   425.1     0.1       0
Bank Sta=247.31,275.81
XS Rating Curve= 0 ,0
Exp/Cntr(USF)=0,0
Exp/Cntr=0.3,0.1

Type RM Length L Ch R = 1 ,15550   ,58.4,59.6,58.8
XS GIS Cut Line= 3
1630407.52526118532203.1698290881630309.23833876532185.248129991
1629980.32361426532244.267176391
#Sta/Elev= 30
       0  825.65    11.3   821.1    17.9  819.04    47.9  812.43    71.3   805.7
    94.6  801.85   144.6   797.5   174.6  797.06     218  797.46   221.3   797.2
  228.48794.6663   234.6  793.59     258  793.07  262.76794.6638     268  797.16
   271.3  797.86   284.5  798.18     298  799.58   311.3   799.5   326.9  807.49
   341.3  813.64     348   818.1   360.8  829.08   374.6  837.24   381.3   842.6
   401.3  865.16   407.9  871.29   411.3  873.89   414.5  875.59   434.1  883.43
#Mann= 4, -1 ,  0
       0    0.06       0  228.48   0.045       0  262.76    0.06       0
  399.91     0.1       0
Bank Sta=228.48,262.76
XS Rating Curve= 0 ,0
Exp/Cntr(USF)=0,0
Exp/Cntr=0.3,0.1

Type RM Length L Ch R = 1 ,15491   ,155.7,154.6,152.2
XS GIS Cut Line= 3
1630404.47279104532145.7464441411630275.16742495532131.906119211
1629977.27114412532186.843791444
#Sta/Elev= 30
       0  821.69    14.7     817    24.6  813.01    70.8  802.52   100.5  801.67
   117.7  798.85   156.8  796.77   196.9  796.06   220.2  796.45   223.6  796.22
  228.08 793.998   230.2  792.89   233.6  792.61  258.37 793.998   290.3  798.21
   310.3  798.54     317  799.82   340.3  812.03     347  817.11   360.3  829.02
     367  833.21   380.4  840.11   383.7  842.51     387  845.66   390.4  849.91
   400.4  863.42     407  870.52   410.4  873.18   420.7  877.78     433  881.05
#Mann= 4, -1 ,  0
       0    0.06       0  228.08   0.045       0  258.37    0.06       0
  390.04     0.1       0
Bank Sta=228.08,258.37
XS Rating Curve= 0 ,0
Exp/Cntr(USF)=0,0
Exp/Cntr=0.3,0.1

Type RM Length L Ch R = 1 ,15336   ,255.5,251.7,239.7
XS GIS Cut Line= 6
1630548.37214686532013.4529106631630255.72760463531964.538222611
1630184.04402097531986.5946089471630088.46612813532016.003342777
1630016.78254447532038.059729114 1629933.1521343532063.792617276
#Sta/Elev= 30
       0  833.79    79.9  812.49    94.2   810.9   110.8  807.74   120.8  807.12
   128.3  805.33   230.9  799.56   348.6  796.83   365.7  794.28   403.5  795.25
  417.91792.6426   423.5  791.06   431.4  790.76  448.33792.6418   454.9   794.9
   465.5  796.38   475.6  796.53   482.4   795.7   485.9  796.22   496.2  801.63
   506.5  809.63   516.8  820.34   523.6  828.54   530.5  833.76   551.1  841.58
   568.2  851.17   585.4  859.58   599.1   864.8   607.2  869.12   634.2  877.29
#Mann= 5, -1 ,  0
       0     0.1       0      80    0.06       0  417.91   0.045       0
  448.33    0.06       0   576.7     0.1       0
Bank Sta=417.91,448.33
XS Rating Curve= 0 ,0
Exp/Cntr(USF)=0,0
Exp/Cntr=0.3,0.1

Type RM Length L Ch R = 1 ,15084   ,390.6,389.9,387
XS GIS Cut Line= 3
1630325.91513375531519.9220178261630109.96075992531703.927920055
1629862.30898073531936.679294731
#Sta/Elev= 30
       0  850.55    44.1  845.42    75.4  839.17   118.5  827.76   142.5  822.61
     182  811.27   213.4  805.11   240.2  798.49   309.9   794.4   353.8  793.24
   372.6  791.55  379.47789.7838   386.5  788.58   406.5  788.99  413.07 789.784
   423.7  792.68   435.3  793.97   468.8  794.93   472.4  795.58     484  801.19
   497.5  806.66   516.5  818.76   547.9  834.76   552.4  836.28   562.9  838.15
   574.9  844.91   597.4  853.67   602.9  856.67     614  865.46   623.6  870.41
#Mann= 7, -1 ,  0
       0     0.1       0      50    0.05       0     130     0.1       0
     170    0.05       0  379.47   0.045       0  413.07    0.06       0
  613.72     0.1       0
Bank Sta=379.47,413.07
XS Rating Curve= 0 ,0
Exp/Cntr(USF)=0,0
Exp/Cntr=0.3,0.1

Type RM Length L Ch R = 1 ,14694   ,339.5,335.5,330.2
XS GIS Cut Line= 2
1629938.23489202531302.7934547061629676.69315052531645.313467353
#Sta/Elev= 30
       0  854.73    61.5  843.72    82.4  836.09   109.9   827.7   115.1  825.14
   143.3  806.62   150.3   802.8   164.4  796.41   172.9   793.5   185.6  791.39
   187.8  790.57  193.63786.0518   197.1  784.62   206.5  784.15   214.2  784.37
  220.42786.0494   225.2  787.14   246.3  789.81   277.5  789.34   284.4  790.55
   313.3  790.08   333.9  791.13   342.2  792.58   354.6  797.19     364  801.63
   379.3  810.81   383.4  812.02   395.8  813.49   428.9  814.12     431  814.86
#Mann= 6, -1 ,  0
       0     0.1       0     190    0.06       0  193.63   0.045       0
  220.42     0.1       0     230    0.06       0     410    0.05       0
Bank Sta=193.63,220.42
XS Rating Curve= 0 ,0
Exp/Cntr(USF)=0,0
Exp/Cntr=0.3,0.1

Type RM Length L Ch R = 1 ,14359   ,271.7,271.5,270.2
XS GIS Cut Line= 2
1629591.32959609531102.4938668461629454.89700822531533.632410115
#Sta/Elev= 30
       0  848.75    20.5  846.86    65.2  844.09    85.8  841.42   103.4  837.72
   120.2  832.68     134  827.43   158.2  821.72   163.5  819.22   168.7  815.45
   171.9  812.13   182.2  798.86   185.6  795.33   189.1  792.69   194.8   785.4
  197.05 783.646   199.4  782.62   202.7  782.29   216.6  782.08     220  782.18
  224.29783.6408   230.4  787.33   233.8  788.03   265.4  787.88   317.7  788.85
   354.3  790.41     370   791.8   381.8  793.75   424.6  806.29   452.2  812.33
#Mann= 7, -1 ,  0
       0     0.1       0      30    0.05       0     120     0.1       0
     170    0.06       0  197.05   0.045       0  224.29    0.06       0
     370    0.05       0
Bank Sta=197.05,224.29
XS Rating Curve= 0 ,0
Exp/Cntr(USF)=0,0
Exp/Cntr=0.3,0.1

Type RM Length L Ch R = 1 ,14087   ,231.6,227.1,222.7
XS GIS Cut Line= 6
1629321.88000375531018.3769090921629300.17105767531103.140847176
1629281.56348334531175.7962136721629256.75382167531272.669707596
1629238.14657542531345.3247460131629216.43631701531430.088356003
#Sta/Elev= 30
       0   797.9    18.7     797    32.5  797.69    42.6  799.06    56.2  802.87
    69.7  805.62    79.9  806.07    86.6  805.35    93.4  803.83     107  797.06
   120.5  794.15   129.5  789.89   134.9  788.37     151  786.85   191.6  786.41
  198.65781.5958   201.8  780.43   208.6  779.81   218.7  779.94   222.1   780.3
  225.93781.5955     232  784.09   235.7  784.86     256  785.16   262.8  785.97
   283.1  785.16   354.2  785.25   391.4  788.53   411.8  791.54     425  795.11
#Mann= 5, -1 ,  0
       0     0.1       0    87.5    0.06       0  198.65   0.045       0
  225.93    0.06       0   357.5    0.05       0
Bank Sta=198.65,225.93
XS Rating Curve= 0 ,0
Exp/Cntr(USF)=0,0
Exp/Cntr=0.3,0.1

Type RM Length L Ch R = 1 ,13860   ,55,55.2,54.9
XS GIS Cut Line= 3
1629036.94651112531001.8768830061629052.98484955531336.978060479
1629071.47201247531468.010529553
#Sta/Elev= 30
       0  799.68    51.3  794.82    54.6  794.06    72.1   787.3    84.1  784.72
   113.7  784.53   130.1  785.84   146.5  784.47     163  784.38   172.8  783.76
   176.1  783.09  183.44 780.306   189.2  778.72   199.1  778.61   212.2  779.15
  216.09780.3055     225  784.03   231.9  784.91   284.5  783.87   340.4  783.64
   377.8  784.27   390.1  784.96   399.3  786.11   416.6  790.13   426.5  793.76
   433.1  796.79   436.5  798.82   449.7  808.96   456.3  815.44   467.8  822.61
#Mann= 7, -1 ,  0
       0     0.1       0      10    0.06       0  183.44   0.045       0
  216.09    0.06       0     310    0.05       0  395.48     0.1       0
  405.48    0.05       0
#XS Ineff= 2 , 0
          159.57  789.27
Permanent Ineff=
       F       F
Bank Sta=183.44,216.09
XS Rating Curve= 0 ,0
Exp/Cntr(USF)=0,0
Exp/Cntr=0.3,0.1

Type RM Length L Ch R = 1 ,13805   ,307,298.9,289.4
XS GIS Cut Line= 2
1628981.72698069531010.427410477 1629005.6409092531468.398308688
#Sta/Elev= 30
       0  801.28    26.3  796.83      46   789.8    65.7  784.95    98.6   783.8
   170.9  783.34   174.1  782.75  181.44779.9348   187.3  778.73   200.4  778.44
   210.3   778.7   213.6  779.38   214.4779.9332   220.1  783.67   223.4  784.52
   246.4  784.07   266.1   784.5   281.7  783.82   361.4  783.12     368  783.31
   377.8  784.81     391  785.06   394.3  785.85   417.3  796.76   420.5  798.92
   427.1  804.73   433.7  809.32   443.5  818.52   450.1  822.17   458.6  825.99
#Mann= 5, -1 ,  0
       0    0.06       0  181.44   0.045       0   214.4    0.06       0
     300    0.05       0     420     0.1       0
#XS Ineff= 2 , 0
          164.26  788.18  300.36          787.85
Permanent Ineff=
       F       F
Bank Sta=181.44,214.4
XS Rating Curve= 0 ,0
Exp/Cntr(USF)=0,0
Exp/Cntr=0.3,0.1

Type RM Length L Ch R = 1 ,13506   ,294.4,290.4,285.2
XS GIS Cut Line= 2
1628613.84482311531160.3124390071628873.01535448531524.142360598
#Sta/Elev= 30
       0  790.26    35.9  789.41    93.9  787.22   118.1  786.98   128.6   786.4
     138  785.29   142.3  783.44     151  777.64   154.5  776.37   166.4   776.1
   174.5  776.44  181.56  777.64   206.2     778   216.8  779.05   230.9  779.88
   273.4  780.05   290.9  780.75   319.5  781.02   335.6  782.59   347.4  782.28
   352.1   783.8   359.1   787.7   371.9  793.75     385  798.88     388     800
   396.8  801.35   409.1  806.44   415.6   807.8   429.7  809.41   446.7  810.26
#Mann= 5, -1 ,  0
       0     0.1       0      30    0.05       0     151   0.045       0
  181.56    0.05       0     250    0.06       0
Bank Sta=151,181.56
XS Rating Curve= 0 ,0
Exp/Cntr(USF)=0,0
Exp/Cntr=0.3,0.1

Type RM Length L Ch R = 1 ,13216   ,321.1,319.7,310.3
XS GIS Cut Line= 2
1628347.26129679531398.0237179621628744.06166443531648.375886743
#Sta/Elev= 30
       0  845.54    20.1  829.91    29.9  823.79    46.3  811.93    60.5  804.28
      76  798.31    97.6  794.12   134.3  780.07   158.1   779.4   169.1  777.13
   180.8  775.83   196.3  775.75   200.2  774.33   205.7  773.03   208.2   773.1
   211.8  774.32   215.7  776.51   223.5  778.03   246.1  776.59   312.7  774.13
   324.3  774.69   332.1  777.24   335.9  777.79   351.5  777.93   368.1  779.08
   386.4  778.69   391.2  781.09     405  792.64   411.1  796.23   469.2  811.99
#Mann= 5, -1 ,  0
       0     0.1       0     180    0.05       0   200.2   0.045       0
   211.8    0.05       0     280    0.06       0
#XS Ineff= 2 , 0
                          371.27          789.59
Permanent Ineff=
       F       F
Bank Sta=200.2,211.8
XS Rating Curve= 0 ,0
Exp/Cntr(USF)=0,0
Exp/Cntr=0.3,0.1

Type RM Length L Ch R = 1 ,12896   ,238.7,240.9,244.5
XS GIS Cut Line= 2
1628180.11961084531717.5550630931628615.98124178531846.580900765
#Sta/Elev= 30
       0  848.86    12.1   847.5    31.7     843    66.9  833.08    79.3  828.89
   102.4  816.47     125  806.37   131.9  800.68     140  792.47     149  781.19
   152.4  778.32   155.8  776.45   162.7  775.12   183.2  775.07   186.6  774.46
  191.37771.9573   193.5  770.59   200.3  769.91  226.39771.9573     238  773.44
   309.8  773.64   326.9  776.76   343.3  778.28   354.3  780.33   378.2  780.72
   382.9  782.81   405.6  799.48   422.5  805.34     433  812.01   454.6  817.99
#Mann= 5, -1 ,  0
       0     0.1       0     140    0.05       0  191.37   0.045       0
  226.39    0.05       0     270    0.06       0
Bank Sta=191.37,226.39
XS Rating Curve= 0 ,0
Exp/Cntr(USF)=0,0
Exp/Cntr=0.3,0.1

Type RM Length L Ch R = 1 ,12655   ,359.3,368,367.3
XS GIS Cut Line= 2
1628147.80605586531920.2193252041628523.11829737532125.655594129
#Sta/Elev= 30
       0  806.85    65.1  795.78      80  790.85    84.8  790.59      95  792.51
   100.4  790.29   106.2  786.12   113.8  776.38   117.4  773.84   128.3   772.2
   141.4  772.53  149.73769.2822   154.8  767.64   158.6  767.62  166.91  769.28
   174.3  772.63   192.2  771.65   215.4  772.11   237.1  769.56   259.6  769.12
   263.7  770.45   270.9  776.73   274.5  778.31   334.4  782.83   353.1  787.75
   371.8  787.44   375.5  788.89   390.5  798.67   401.5   803.1   427.9  817.36
#Mann= 5, -1 ,  0
       0     0.1       0      60    0.06       0  149.73   0.045       0
  166.91    0.06       0     400     0.1       0
Bank Sta=149.73,166.91
XS Rating Curve= 0 ,0
Exp/Cntr(USF)=0,0
Exp/Cntr=0.3,0.1

Type RM Length L Ch R = 1 ,12287   ,302.7,322.7,329.2
XS GIS Cut Line= 3
1627986.54701408532071.6702876351628017.93522478532181.177762942
1628314.68934242532443.433114661
#Sta/Elev= 30
       0  798.17    15.5  795.49      36  790.55    53.3  785.07    66.5  778.69
    74.5  777.09    87.2  771.99   149.4  772.25   232.8  769.03   253.7   769.2
  273.46 765.332   281.6  763.75   293.1  763.59   302.5  764.27  305.63765.3308
   307.9  766.71   319.6  779.09   332.7  786.26   337.6  788.03   342.6  788.55
   351.3  788.61   360.6  787.46   376.5  797.48   394.1  803.42   421.9  816.78
   426.8  820.02   459.7  846.15   476.4  853.82   496.2  866.21   509.9  872.45
#Mann= 5, -1 ,  0
       0     0.1       0     110    0.06       0  273.46   0.045       0
  305.63    0.06       0  373.92     0.1       0
Bank Sta=273.46,305.63
XS Rating Curve= 0 ,0
Exp/Cntr(USF)=0,0
Exp/Cntr=0.3,0.1

Type RM Length L Ch R = 1 ,11965   ,274.4,277.2,275.2
XS GIS Cut Line= 2
1627841.53453867532073.0593637721627852.52864248532571.955584398
#Sta/Elev= 30
       0  798.89     9.2  797.93    29.9   793.3      43  786.83    62.7  773.71
      66  772.01    72.6  770.46    98.8  768.81   207.1  769.21   233.4  767.71
   243.2  766.28   259.6  766.44   266.2  765.34  271.58763.0974     299  761.62
  307.61763.0955   312.1   765.7   325.2     776   328.5  777.35   344.9   778.2
   348.2  780.71   354.8  790.97   358.1   794.7   367.9  803.79   374.5  808.75
   390.9  817.32   420.2  827.74   440.1  832.24   472.9  844.77     499  852.52
#Mann= 6, -1 ,  0
       0     0.1       0     130    0.05       0     220    0.06       0
  271.58   0.045       0  307.61    0.06       0     430     0.1       0
Bank Sta=271.58,307.61
XS Rating Curve= 0 ,0
Exp/Cntr(USF)=0,0
Exp/Cntr=0.3,0.1

Type RM Length L Ch R = 1 ,11687   ,306.3,301,286.2
XS GIS Cut Line= 6
  1627578.616758532147.596763507 1627575.2683395532235.096588507
1627573.72798826532310.0967665911627573.72798826532410.096566588
1627573.72798826532485.0967446711627573.72798826532572.596569672
#Sta/Elev= 30
       0  815.87    24.3  807.49    36.4  801.56      44  797.04    57.1   785.8
    70.2  776.11    83.4  770.91   103.1   767.5   116.2  766.01   145.7  764.15
   175.3  764.01  190.99760.5919   198.2   759.4   211.3  759.24   221.2   759.4
   224.5  759.79  226.35760.5936   234.3  765.03   237.6  766.13   240.9  766.56
     254  767.05   290.1   767.1   329.5  768.61   352.4  770.69   355.7  771.26
   363.5  773.74   368.8  774.49   381.9  774.59   391.8  773.75   425.1  780.29
#Mann= 3, -1 ,  0
       0     0.1       0  190.99   0.045       0  226.35    0.06       0
Bank Sta=190.99,226.35
XS Rating Curve= 0 ,0
Exp/Cntr(USF)=0,0
Exp/Cntr=0.3,0.1

Type RM Length L Ch R = 1 ,11386   ,288,299,289.2
XS GIS Cut Line= 4
 1627211.2190487532275.1863143671627296.90603533532400.067715257
1627366.33798309532472.7673730111627504.65681219532655.196796728
#Sta/Elev= 30
       0  873.37    24.5  859.22    29.9  855.28    33.8  853.72    43.4  851.55
      63  839.95    81.6  830.42    93.5  820.75   105.5   812.9   109.4  808.84
   125.3  788.63   144.2  772.22     158  764.52   165.8  758.37   171.6  757.25
  181.66  757.08     193  756.53  208.09  757.08     212  758.33   216.8   761.3
   219.2  762.12   235.8   764.3   335.5  766.13   380.5  771.03   389.8  773.03
   403.9  773.47   413.7  772.44   422.6  774.27   456.1     776   480.9  778.26
#Mann= 5, -1 ,  0
       0     0.1       0  181.66   0.045       0  208.09    0.05       0
  251.45    0.06       0  480.92    0.05       0
Bank Sta=181.66,208.09
XS Rating Curve= 0 ,0
Exp/Cntr(USF)=0,0
Exp/Cntr=0.3,0.1

Type RM Length L Ch R = 1 ,11087   ,289.9,300,307.2
XS GIS Cut Line= 6
1626966.77250926532442.9997159991627023.64772359532509.494005591
1627072.39795418 532566.488642261627137.39815226532642.481928587
1627186.14838284532699.4768933361627243.02359718532765.970854834
#Sta/Elev= 30
       0  831.34    18.8  819.71    22.6   816.5      25  815.12    27.4  813.99
    36.1  812.74    41.3  811.03    62.5  799.79    83.6  786.99   113.8   774.1
     125  766.57   129.7  764.25   134.3  762.91     144  761.33   183.6  760.14
   187.9  759.24  198.74754.1784   204.1   753.1   208.9  752.85     224  753.24
   234.1754.1782   241.4  756.35   255.3  762.11   259.3  762.85   314.9  766.73
   329.6  769.09   351.2  768.98   359.9  771.31   394.4  775.82     425   778.3
#Mann= 5, -1 ,  0
       0     0.1       0   137.5    0.06       0  198.74   0.045       0
   234.1    0.06       0   357.5    0.05       0
Bank Sta=198.74,234.1
XS Rating Curve= 0 ,0
Exp/Cntr(USF)=0,0
Exp/Cntr=0.3,0.1

Type RM Length L Ch R = 1 ,10787   ,287.6,288.5,288.8
XS GIS Cut Line= 6
1626811.85484008532550.6336870941626830.35775584532636.177479252
1626844.76028609532709.7911771681626864.06241284532807.910731584
1626878.46133417532881.5060568451626895.26149742532967.373011082
#Sta/Elev= 30
       0   801.5    18.6  790.08    42.1  782.03    61.1  771.03    69.4  767.28
    92.4   762.4   102.5  760.96   129.2  758.94   175.4  756.84  191.22751.7747
   196.1  750.79   212.8  749.96   219.5  750.34  223.83751.7775   229.5  756.35
   232.9  758.11   236.2   758.6   289.7  758.93   306.4  758.27   316.4  759.06
   323.1  760.92   326.5   762.7   329.8  765.81   336.5  775.25   339.8   778.7
   366.6  797.03   376.6  804.79     390   813.5     413  822.75     425  830.41
#Mann= 5, -1 ,  0
       0     0.1       0  137.52    0.06       0  191.22   0.045       0
  223.83    0.06       0  322.53     0.1       0
Bank Sta=191.22,223.83
XS Rating Curve= 0 ,0
Exp/Cntr(USF)=0,0
Exp/Cntr=0.3,0.1

Type RM Length L Ch R = 1 ,10499   ,312.7,309,304
XS GIS Cut Line= 6
1626547.54616403532635.3870957881626557.79450312532722.375110784
1626568.40832704532796.6361171251626584.58644428532895.318662533
1626596.71995021532969.3306536171626610.87543371533055.677921871
#Sta/Elev= 30
       0  808.24    11.5  804.97    28.8  797.82      42   793.2    71.7  781.06
    88.2  773.04   104.8  767.31   121.4  757.67   131.3  756.05   141.3  755.82
   144.6  754.72   151.2   750.7  153.44 750.028   161.2  748.63   171.1  748.41
   181.1  748.82  185.43750.0251   197.7  754.36     211  756.17   240.9  756.36
   254.2  755.52   297.5  754.91   330.7  756.33   347.3  755.91   350.7  756.74
     364  762.09   376.4  768.56   387.2  772.75   397.2  777.83   425.1  787.38
#Mann= 5, -1 ,  0
       0     0.1       0  153.44   0.045       0  185.43     0.1       0
  202.61    0.06       0  387.61     0.1       0
#XS Ineff= 2 , 0
                          239.35          759.65
Permanent Ineff=
       F       F
Bank Sta=153.44,185.43
XS Rating Curve= 0 ,0
Exp/Cntr(USF)=0,0
Exp/Cntr=0.3,0.1

Type RM Length L Ch R = 1 ,10190   ,300.2,302.5,299.4
XS GIS Cut Line= 6
1626235.13528141532792.538146168 1626271.2277289532872.197435661
1626302.16401875 532940.477810921626345.27220024533030.969755917
1626380.29936115533100.1435020871626424.60340641533180.196819662
#Sta/Elev= 30
       0   812.2     6.5   809.6    24.5  799.62    30.2  796.89    46.1  789.91
    60.6  784.96    67.8  781.29    71.4  778.67    74.9  774.76    78.6  767.17
    82.3  758.09    84.8   753.6    87.2  750.62   90.43748.2433    94.7  746.99
   104.6  746.63   118.2  746.81   121.8  747.35  123.89748.2423     129  750.33
   132.6   750.8   172.3  752.51   299.9  753.09     333  754.77   374.1  755.52
   391.3  757.49   408.9  757.29   413.1   758.5   422.4  764.64   431.7  769.52
#Mann= 4, -1 ,  0
       0     0.1       0   90.43   0.045       0  123.89     0.1       0
  182.42    0.06       0
#XS Ineff= 2 , 0
                          254.51          755.98
Permanent Ineff=
       F       F
Bank Sta=90.43,123.89
XS Rating Curve= 0 ,0
Exp/Cntr(USF)=0,0
Exp/Cntr=0.3,0.1

Type RM Length L Ch R = 1 ,9887    ,566.1,600.6,627.2
XS GIS Cut Line= 6
1625939.55277893 532896.968296261625986.93063693532970.818870336
1626023.35477668533036.3800909221626071.91799976533123.796582758
1626108.34082717533189.3584595021626150.83385243 533265.84780784
#Sta/Elev= 30
       0  805.11      35  807.61      51  805.32    72.3  800.01    81.8  798.45
    96.2  794.62   108.3  789.56   121.8  785.18     127  782.32   130.8  779.72
   134.6   776.5   138.3  772.48   144.5     765   148.8  760.95   160.8   752.9
   164.6  750.71   175.8   748.5  184.92745.9565   194.6  745.03   209.6  744.72
   220.9  745.02  227.46745.9571   233.7  747.51   239.6  748.37   265.9  750.07
   318.5  750.67   329.7  751.42   352.2  752.14   398.8  751.66   425.2  752.06
#Mann= 4, -1 ,  0
       0     0.1       0  182.74    0.06       0  184.92   0.045       0
  227.46    0.06       0
Bank Sta=184.92,227.46
XS Rating Curve= 0 ,0
Exp/Cntr(USF)=0,0
Exp/Cntr=0.3,0.1

Type RM Length L Ch R = 1 ,9287    ,259.1,271,279.2
XS GIS Cut Line= 6
1625909.86718824532913.5217610911625681.63512627532978.143877879
1625589.83956759533026.9772225921625501.09269784533073.080804929
1625434.12104701533106.8445169181625355.98832926533146.235186175
#Sta/Elev= 30
       0  792.73    11.8  787.68    39.1  778.55    59.6  769.62    66.4  765.67
    76.6  756.21    83.4  750.97    93.7  747.32   148.2  744.76   280.8  745.87
   294.8  742.75   348.3  744.22   359.4  741.19   371.1  741.67     376740.4275
   381.6  739.12   403.8  738.73  411.41740.4235   414.8   742.9   422.2  751.14
   429.6  756.31   441.6  757.66   455.4  757.34   458.7  758.38   470.1  765.72
   495.4  774.61   536.3  793.52     562  810.27   581.9   818.1   603.7   832.2
#Mann= 7, -1 ,  0
       0     0.1       0     220    0.05       0   247.2     0.1       0
   317.2    0.06       0     376   0.045       0  411.41    0.06       0
  526.19     0.1       0
#XS Ineff= 2 , 0
          234.01  751.84
Permanent Ineff=
       F       F
Bank Sta=376,411.41
XS Rating Curve= 0 ,0
Exp/Cntr(USF)=0,0
Exp/Cntr=0.3,0.1

Type RM Length L Ch R = 1 ,9016    ,232.4,224.5,215.4
XS GIS Cut Line= 2
1625872.73657613532819.5165000971625427.55711042532782.066263791
#Sta/Elev= 30
       0  779.42     7.1  778.25    13.7   775.6    30.1  763.82      40  757.67
    46.6  754.67    63.1  749.16    79.5  746.47      96  741.91   125.6  742.89
   158.5  741.57   168.4  742.41   194.8     743   224.4  741.57   247.4  742.04
   316.6   741.6   326.7  742.18  351.14738.3912   379.1  736.47   385.7  737.36
  386.89738.3938   392.3  744.13   395.6  746.79   398.9  747.99   418.6   748.5
   421.9  750.15   428.5  759.15   435.1  767.13   441.7  773.12   446.8  776.76
#Mann= 6, -1 ,  0
       0     0.1       0     210    0.05       0     270     0.1       0
  351.14   0.045       0  386.89     0.1       0     390    0.06       0
Bank Sta=351.14,386.89
XS Rating Curve= 0 ,0
Exp/Cntr(USF)=0,0
Exp/Cntr=0.3,0.1

Type RM Length L Ch R = 1 ,8791    ,306.8,310.4,293.4
XS GIS Cut Line= 2
1625822.04099338532495.4767051591625417.43126728532607.124176483
#Sta/Elev= 30
       0  777.65     5.8  775.72    26.2  767.16    39.8  758.93    53.4  752.17
    90.9  742.03    97.7  740.72   148.7  739.17   189.6  741.19   203.2  738.61
     244  740.03   250.8  739.56   257.5736.7559     261  735.97   271.3  735.43
   295.1  735.63  304.38736.7576   322.3  740.24   335.9  741.29   344.7  744.24
   349.5  745.19   359.7  745.56     370  744.85   373.4  745.78   383.6  750.45
     387  753.43   390.4  758.48   393.8  762.62   405.6  771.76   419.7  779.39
#Mann= 3, -1 ,  0
       0     0.1       0   257.5   0.045       0  304.38    0.06       0
Bank Sta=257.5,304.38
XS Rating Curve= 0 ,0
Exp/Cntr(USF)=0,0
Exp/Cntr=0.3,0.1

Type RM Length L Ch R = 1 ,8481    ,68.3,72.4,68.2
XS GIS Cut Line= 6
1625607.43400897532167.7026097991625553.90032337532237.360278882
1625504.64025129532294.114102385 1625437.0655833532368.152012057
1625386.77270488532423.8100372181625328.74034063532489.337793313
#Sta/Elev= 30
       0  762.87    12.3  762.25      20  761.03    62.1  750.12    75.6  747.15
   117.7  740.12   127.7  739.41   167.7  739.84   171.6  739.13  180.04734.8439
     184  733.57   192.5  733.09   210.7  733.74  215.85734.8433     225  737.05
   250.7  737.64   260.1  736.92   277.2   737.3   292.3  738.71   304.1  741.06
   325.9  742.03   343.4   749.3   359.7   759.9     378  768.53   382.9  770.68
   397.8  774.91   407.7  778.89   412.6  782.57   417.8  787.73   425.8  792.82
#Mann= 4, -1 ,  0
       0     0.1       0      50    0.06       0  180.04   0.045       0
  215.85    0.06       0
#XS Ineff= 2 , 0
          165.35  747.41
Permanent Ineff=
       F       F
Bank Sta=180.04,215.85
XS Rating Curve= 0 ,0
Exp/Cntr(USF)=0,0
Exp/Cntr=0.3,0.1

Type RM Length L Ch R = 1 ,8408    ,328.3,319.6,310.5
XS GIS Cut Line= 5
1625587.19507771532155.6093089491625469.28511941532231.633466128
1625396.67171788532311.7178560481625346.37883946532367.375881209
1625288.34647521532432.903637304
#Sta/Elev= 30
       0  758.62    16.8  756.05    43.4  748.71    76.1  742.52      88  742.01
    94.2  740.89   113.7   740.2   126.8  738.67   133.2  738.75   141.2  740.62
   149.5  738.67  179.35 734.425   192.5  733.14   205.7  732.84   214.6  733.04
  219.87 734.425   223.8  736.36   228.5  737.26   272.6  737.33   287.8  739.26
   311.9  739.16   314.4  739.68   317.1  740.98   328.3   750.4   346.9  763.33
   356.7  767.71   367.9  771.68   391.3  777.86   398.1  781.24   410.9  790.73
#Mann= 5, -1 ,  0
       0     0.1       0      40    0.06       0  179.35   0.045       0
  219.87    0.06       0  383.41     0.1       0
Bank Sta=179.35,219.87
XS Rating Curve= 0 ,0
Exp/Cntr(USF)=0,0
Exp/Cntr=0.3,0.1

Type RM Length L Ch R = 1 ,8089    ,632.1,625.9,598
XS GIS Cut Line= 4
1625215.15330938531901.0416023191625136.84679673 532189.32672633
1625120.22511082532262.4617506681625100.83407348532347.786055085
#Sta/Elev= 30
       0  744.43    73.2  739.73   103.8  738.86   120.8  737.35   134.4  737.28
   168.4   734.9   195.6  734.22   209.2  734.47  216.87 732.469   222.8   731.4
   236.4  730.84   246.6  730.91  253.44732.4672   256.8  733.51   260.2  733.69
   273.8   733.2   280.6  733.98   290.8  736.17   351.5  735.83   358.2  736.38
   368.3  739.13     375  739.88   385.1  740.19   398.6  739.18   408.7  742.42
   420.8  744.15   438.9  748.32   445.7  751.31   455.8  757.22   461.2  759.69
#Mann= 4, -1 ,  0
       0     0.1       0  216.87   0.045       0  253.44     0.1       0
     290    0.06       0
Bank Sta=216.87,253.44
XS Rating Curve= 0 ,0
Exp/Cntr(USF)=0,0
Exp/Cntr=0.3,0.1

Type RM Length L Ch R = 1 ,7463    ,279.6,283.9,286.2
XS GIS Cut Line= 5
1624587.11006344532070.3243672041624647.61322327532133.534870707
 1624699.4726996 532187.716192791624769.83673209532258.791838043
1624904.47506265 532452.00160304
#Sta/Elev= 30
       0  776.81    22.3  770.98    27.1  768.92    31.7  765.89    46.1  753.04
    66.5  731.16    68.8  728.79   70.89727.3644      77  726.14    87.5  726.49
    98.3  726.03   103.6  726.29  108.73727.3627   117.2  730.02   126.9  731.44
   172.5  730.74   212.7  731.39   279.8  733.68   324.5  733.86   348.5  735.06
   374.5  735.52   416.9  737.86   423.3     739   428.7  741.79   432.5  742.74
   452.5  743.38   463.4  747.52   469.2  748.93   480.5  750.98     498  752.77
#Mann= 5, -1 ,  0
       0     0.1       0   70.89   0.045       0  108.73     0.1       0
   232.5    0.05       0  342.51    0.06       0
Bank Sta=70.89,108.73
XS Rating Curve= 0 ,0
Exp/Cntr(USF)=0,0
Exp/Cntr=0.3,0.1

Type RM Length L Ch R = 1 ,7179    ,292,290.4,286.6
XS GIS Cut Line= 2
1624333.61218186532164.5555707011624633.60928586532583.853762406
#Sta/Elev= 30
       0  806.03      17  799.49      24  794.89    39.3  781.57    49.3  777.01
    66.3  771.85    80.4  763.23    89.8  754.19    92.2  752.72     107  749.19
   113.9  745.14     126  736.22     134  731.95   150.2  729.68   182.4  729.39
   186.5  728.65  194.58725.0894   202.7  723.91   225.4  723.78   234.9  724.01
  239.85725.0904   247.4  729.18   259.1  730.56   331.7  731.69   388.2  733.75
     412  736.47   440.6   742.1   463.7  748.63     489  749.05   515.6  761.06
#Mann= 4, -1 ,  0
       0     0.1       0  194.58   0.045       0  239.85     0.1       0
     380    0.06       0
Bank Sta=194.58,239.85
XS Rating Curve= 0 ,0
Exp/Cntr(USF)=0,0
Exp/Cntr=0.3,0.1

Type RM Length L Ch R = 1 ,6889    ,390.5,402.8,406.7
XS GIS Cut Line= 6
1624101.69424993532364.5549910071624157.69249751532432.075197175
1624205.94272909532489.7082840061624273.25853933 532563.70026201
1624325.10029918532617.8983163391624385.58180551532681.130145252
#Sta/Elev= 30
       0  782.48    13.7  780.55    58.1  776.54    76.7  773.22    80.5  771.15
    83.7  768.22   103.5  745.16     112  736.61   120.6  729.13   124.9  727.09
   130.3  726.29     142  727.16   181.9  727.71   186.7  727.04  192.77723.6627
   196.5  722.39   201.4  722.12   225.7  722.19   230.3  722.54  234.41723.6638
   239.5  725.46   251.2  726.66   260.4  728.89   292.7  729.68   320.8  731.34
     344  734.57     379  737.61   392.7  741.06   415.3  741.82   425.4  743.96
#Mann= 4, -1 ,  0
       0     0.1       0  192.77   0.045       0  234.41     0.1       0
  347.92    0.06       0
Bank Sta=192.77,234.41
XS Rating Curve= 0 ,0
Exp/Cntr(USF)=0,0
Exp/Cntr=0.3,0.1

Type RM Length L Ch R = 1 ,6486    ,258.1,274.3,279.1
XS GIS Cut Line= 3
1623830.92427258 532464.315470161623838.41707957532564.991496237
1623999.47893592532955.220682986
#Sta/Elev= 30
       0  757.32    22.6   753.6    52.2  746.81    59.2  743.98    80.5  732.74
    88.4  730.76   140.6   727.6   172.5  727.22   176.1  726.67   184.1  723.52
   190.3  722.72   200.9   724.5   211.7  724.97   237.8  724.52   254.2  721.94
   282.6   721.7   289.7  720.93   321.6  720.05   325.2  720.33  329.38721.6889
   334.8  725.78   339.4  727.02     370  728.33   381.9  728.19   399.7  732.39
   438.7  745.85     460  754.74   483.3  760.08   499.1  764.49   523.1  773.92
#Mann= 5, -1 ,  0
       0     0.1       0  230.95    0.06       0   282.6   0.045       0
  329.38    0.06       0  430.95     0.1       0
Bank Sta=282.6,329.38
XS Rating Curve= 0 ,0
Exp/Cntr(USF)=0,0
Exp/Cntr=0.3,0.1

Type RM Length L Ch R = 1 ,6212    ,533.5,522.6,516.3
XS GIS Cut Line= 2
 1623672.9610667532480.4279420471623646.56398687532989.282982701
#Sta/Elev= 30
       0  753.99     9.7  750.92    26.1  743.41    49.1  738.52    55.7  735.42
    65.5  729.43    72.1  727.64   200.2  723.86   269.2  723.64   275.8  722.68
  280.52720.2223   285.6  718.49   292.1  718.16  325.48720.2227   331.6  724.64
   334.9  726.22   354.6  727.37   357.9  728.85   361.2  731.33   380.9  753.87
   384.2  758.16   397.3   778.2   403.9     786   407.2  788.71   423.6  797.08
   433.5  803.12   441.1  806.67   453.2  814.12   495.9  831.73   509.5  838.42
#Mann= 5, -1 ,  0
       0     0.1       0     270    0.06       0  280.52   0.045       0
  325.48    0.06       0     450     0.1       0
Bank Sta=280.52,325.48
XS Rating Curve= 0 ,0
Exp/Cntr(USF)=0,0
Exp/Cntr=0.3,0.1

Type RM Length L Ch R = 1 ,5689    ,329.9,317.6,304.7
XS GIS Cut Line= 3
1623091.71902708532504.4248792671623128.51550961532586.266148964
1623437.34136327533062.918002279
#Sta/Elev= 30
       0  766.31    27.6  763.21    52.6  758.33    84.7  755.16    97.5  752.54
   121.7  745.88   137.1  739.27   157.9  733.74   178.4  724.12  189.75716.6331
   194.1   715.5   209.7  715.07  222.05716.6326   229.6   718.5   248.8  718.92
   266.5  721.58   281.8  720.51   334.8  720.22     372  721.26   478.7  721.19
   514.6  722.22   519.1   723.5     538  732.78   553.7  734.52   592.8  735.82
   597.3  737.84   610.4  747.07   622.5  752.87   634.5  762.32   657.7  775.31
#Mann= 6, -1 ,  0
       0     0.1       0  189.75   0.045       0  222.05     0.1       0
  249.73    0.07       0  459.73    0.06       0  579.73     0.1       0
#XS Ineff= 2 , 0
                          403.32          724.37
Permanent Ineff=
       F       F
Bank Sta=189.75,222.05
XS Rating Curve= 0 ,0
Exp/Cntr(USF)=0,0
Exp/Cntr=0.3,0.1

Type RM Length L Ch R = 1 ,5371    ,311.1,302,293
XS GIS Cut Line= 3
1622853.70554331532873.1971667321623144.19156951532971.449335189
 1623354.8925606533132.986282719
#Sta/Elev= 30
       0  755.81    11.1  749.25    31.4   741.9    41.8  737.32    59.1  728.82
    72.9  723.41    79.9  721.62    90.2  720.14   124.9  717.41  132.86713.8343
   138.7  713.02   169.9  712.51   173.4  712.71  177.89713.8339   197.4  716.96
     260  718.55   273.8  718.97   291.1  720.45   329.5  721.03   392.8  720.01
   416.3  720.56   430.2  719.96   445.2  722.08   474.2  728.34   491.5  730.84
   502.7   733.4   516.8  735.12   547.2  743.19   561.6  744.57   572.2  744.85
#Mann= 8, -1 ,  0
       0     0.1       0  132.86   0.045       0  177.89     0.1       0
     190    0.06       0     260    0.07       0  506.65    0.06       0
  526.65    0.07       0  546.65     0.1       0
Bank Sta=132.86,177.89
XS Rating Curve= 0 ,0
Exp/Cntr(USF)=0,0
Exp/Cntr=0.3,0.1

Type RM Length L Ch R = 1 ,5069    ,122.8,123.8,126.3
XS GIS Cut Line= 4
1622707.80823717533142.5184245921622857.19013009533212.751874557
1622981.45201752533203.939689454 1623184.9473722533241.885504912
#Sta/Elev= 30
       0  753.49    16.4     751    30.9  747.94    56.3  745.48    92.9  739.34
   147.1  728.06   150.6  727.26   154.2   725.9   165.1  719.03   168.3  717.63
   174.9  715.97   181.5  714.95   184.8  714.04  190.72711.6096   194.7   710.7
   197.9  710.54   224.3  710.28   234.1  710.74  237.53711.6085   250.6  716.13
   253.9  716.62   276.9  717.69   299.6  719.34   336.8  720.36   370.1  722.62
   400.2  723.81   413.5  725.56   420.2  725.63   450.2  728.23   496.6  731.11
#Mann= 5, -1 ,  0
       0     0.1       0     130    0.06       0  190.72   0.045       0
  237.53    0.06       0  255.07    0.07       0
Bank Sta=190.72,237.53
XS Rating Curve= 0 ,0
Exp/Cntr(USF)=0,0
Exp/Cntr=0.3,0.1

Type RM Length L Ch R = 1 ,4945    ,133.7,152.3,162.6
XS GIS Cut Line= 4
1622671.86653948533241.5975564881622827.96674379533327.507066358
1622942.15116414533325.413192642  1623122.068605 533375.24817982
#Sta/Elev= 30
       0  733.41     5.8  732.23      13  731.24    40.4  728.58    51.7  725.65
    65.5  723.98      88  719.56   101.6  717.76   108.4  716.42   122.1  717.33
   135.7  717.52   153.2  716.11   177.8  714.98   187.1  713.64  194.71710.8631
   197.6  710.18   207.4   709.4     214  709.25   230.4  709.63  237.32 710.862
   243.1  712.55   250.1  715.23   253.3  716.04   259.9  716.98   266.5  717.18
   296.1  716.81   316.6  717.33   358.6  720.21   421.7  722.91   479.1  726.17
#Mann= 5, -1 ,  0
       0     0.1       0      90    0.06       0  194.71   0.045       0
  237.32    0.06       0  422.38    0.05       0
Bank Sta=194.71,237.32
XS Rating Curve= 0 ,0
Exp/Cntr(USF)=0,0
Exp/Cntr=0.3,0.1

Type RM Length L Ch R = 1 ,4793    ,385.8,395.9,402.1
XS GIS Cut Line= 4
1622615.37184722533271.7650904351622841.02485526533497.214471087
1622896.96929717533547.1667990091622960.19554867533607.731310427
#Sta/Elev= 30
       0  730.43    12.7   727.4    26.7  722.55    40.6  719.47    49.8  717.95
    61.4  717.04    68.4  715.96   138.1  715.31   158.8   714.3   170.6   712.9
   188.9  713.88   207.3  713.51   219.1  712.93   226.3  711.41   237.7  710.96
  250.11709.2015   263.4  707.65   274.8  708.28  278.49709.2023   286.6  714.54
   314.2  715.47   358.5   715.6   367.7  716.08   378.2  717.48   388.1  719.44
     412   726.2   423.4  728.61   434.3  729.92   466.1  732.41   481.5  734.43
#Mann= 5, -1 ,  0
       0     0.1       0      60    0.06       0  250.11   0.045       0
  278.49    0.06       0  378.98    0.05       0
Bank Sta=250.11,278.49
XS Rating Curve= 0 ,0
Exp/Cntr(USF)=0,0
Exp/Cntr=0.3,0.1

Type RM Length L Ch R = 1 ,4397    ,217.6,221,221.3
XS GIS Cut Line= 3
1622414.18175293533277.9586967021622424.74985443 533492.91056025
1622506.40449382533830.523318125
#Sta/Elev= 30
       0  727.52     9.4  723.77    15.9  722.04    65.2  720.82    84.9  718.73
   111.2  713.86   124.3   714.4   147.3  713.88   206.5  714.59     240  714.22
   253.6  713.24   304.1  711.81   338.1  711.84   341.2  711.64   343.3  710.74
  348.08 707.181   351.5  705.54   361.5  704.77   371.6  705.15  379.58 707.184
   424.9  710.48   439.1  716.44   446.6  717.72   472.9   719.8   489.8   720.2
   503.3  722.35   523.5  726.58     537  730.28   547.2  733.97   562.6  741.44
#Mann= 3, -1 ,  0
       0    0.06       0  348.08   0.045       0  379.58     0.1       0
Bank Sta=348.08,379.58
XS Rating Curve= 0 ,0
Exp/Cntr(USF)=0,0
Exp/Cntr=0.3,0.1

Type RM Length L Ch R = 1 ,4176    ,277.2,284.1,290.4
XS GIS Cut Line= 5
1622208.79299023533276.615890382 1622248.9748531533548.428479656
1622267.50801192533691.4146040181622274.96961117533766.042735602
1622283.67497434533853.108506361
#Sta/Elev= 30
       0  721.68    37.4  718.03    63.3  717.52    71.9  717.04    80.5  715.88
    97.1  715.59   126.8  713.88     170  712.19   223.1  711.78   278.7   713.1
   305.9  711.77   345.6  710.91   372.1   710.7   405.2  711.11   420.6  709.68
   434.9  709.59   444.8  706.91  454.41705.7275   461.3  704.75   467.9  704.38
     481  704.58  484.29705.7261   490.9  712.14   498.6  718.51   507.4  726.64
     514  731.21   525.5  736.96   553.6  749.58   573.4  756.94   581.4  760.37
#Mann= 6, -1 ,  0
       0     0.1       0     100    0.07       0     190    0.06       0
  404.77     0.1       0  454.41   0.045       0  484.29     0.1       0
Bank Sta=454.41,484.29
XS Rating Curve= 0 ,0
Exp/Cntr(USF)=0,0
Exp/Cntr=0.3,0.1

Type RM Length L Ch R = 1 ,3892    ,304,307.7,310.9
XS GIS Cut Line= 4
1622091.16292704533341.5271455661622058.80352339533499.875835917
1621979.69915009533727.3232628411621957.64243567533799.006518424
#Sta/Elev= 30
       0   716.7    95.4  711.83   132.2  710.57   148.9   709.4     159  710.24
   169.3  710.16   231.8  708.12   294.4  708.33   321.1  707.77   329.1  706.94
   332.6  705.78  336.83703.3174   339.5  702.19   353.4  701.53   363.8  701.75
   367.5  702.27  370.02 703.319   374.3   706.7   377.6  711.56   381.2  716.06
   402.4  735.96   408.8  739.67   415.8  742.65   427.2  748.85   443.2  755.33
   446.7  757.26     457   765.6   464.3  769.99   467.3  772.38   477.4  782.99
#Mann= 4, -1 ,  0
       0    0.06       0  311.62     0.1       0  336.83   0.045       0
  370.02     0.1       0
Bank Sta=336.83,370.02
XS Rating Curve= 0 ,0
Exp/Cntr(USF)=0,0
Exp/Cntr=0.3,0.1
